--- TENMILECK.prj (project) ---

Proj Title=TENMILECK
Current Plan=p01
Default Exp/Contr=0,0
English Units
Geom File=g01
Flow File=f01
Plan File=p01
BEGIN DESCRIPTION:
-------- MODELED AS PART OF WVEMD CTP PROGRAM, 2023----------
Stream Name: Tenmile Creek
Flood Zone:  AFH
Upshur County, WV
HEC-RAS Version: RAS 6.3
Vertical Datum: NAVD88
Projection: NAD 1983 StatePlane West Virginia S FIPS 4702 (US Feet)
Terrain: 1-meter LIDAR (FEMA Region III 3DEP collected 2016-2018)
Land Use: 2019 NLCD
Hydrologic Method:
WV SIR2010-5033 regression equations
Additional Model Notes:
None
END DESCRIPTION:
DSS Export Rating Curves= 0
DSS Export Rating Curve Sorted= 0
DSS Export Volume Flow Curves= 0
DXF OffsetX= 0
DXF OffsetY= 0
DXF ScaleX= 0
DXF ScaleY= 0

--- TENMILECK.p01 (plan) ---

Plan Title=Floodplain
Program Version=6.31
Short Identifier=Floodplain
Geom File=g01
Flow File=f01
Subcritical Flow
K Sum by GR= 0
Std Step Tol= 0.01
Critical Tol= 0.01
Num of Std Step Trials= 20
Max Error Tol= 0.3
Flow Tol Ratio= 0.001
Split Flow NTrial= 30
Split Flow Tol= 0.02
Split Flow Ratio= 0.02
Log Output Level= 0
Friction Slope Method= 1
Unsteady Friction Slope Method= 2
Unsteady Bridges Friction Slope Method= 1
Parabolic Critical Depth
Global Vel Dist= 0 , 0 , 0
Global Log Level= 0
CheckData=True
Encroach Param=-1 ,0,0, 0
Mapping Interval=1HOUR
Computation Time Step Use Courant=        0
Computation Time Step Use Time Series=    0
Computation Time Step Count To Double=0
Computation Time Step Max Doubling=0
Computation Time Step Max Halving=0
Computation Time Step Residence Courant=0
Run HTab= 0
Run UNet= 0
Run Sediment= 0
Run PostProcess= 0
Run WQNet= 0
Run RASMapper=-1
UNET Theta= 0
UNET Theta Warmup= 0
UNET ZTol= 0
UNET ZSATol= 0
UNET MxIter= 0
UNET Max Iter WO Improvement= 0
UNET MaxInSteps= 0
UNET DtIC= 0
UNET DtMin= 0
UNET MaxCRTS= 0
UNET WFStab= 0
UNET SFStab= 0
UNET WFX= 1
UNET SFX= 1
UNET Gravity=32.17405
UNET 1D Methodology=Finite Difference
UNET DSS MLevel= 1
UNET Pardiso=0
UNET DZMax Abort= 0
UNET Use Existing IB Tables= 0
UNET Froude Reduction=False
UNET Froude Limit= 0
UNET Froude Power= 0
UNET D1 Cores= 0
UNET WindReference=Eulerian
UNET WindDragFormulation=Hsu (1988)
UNET D2 Coriolis=0
UNET D2 Cores= 0
UNET D2 Theta= 1
UNET D2 Theta Warmup= 1
UNET D2 Z Tol= 0.01
UNET D2 Volume Tol= 0.01
UNET D2 Max Iterations= 20
UNET D2 Equation= 0
UNET D2 RampUpFraction=0.1
UNET D2 TimeSlices= 1
UNET D2 Turbulence Formulation=Non-Conservative (original)
UNET D2 Eddy Viscosity=0.3
UNET D2 Transverse Eddy Viscosity=0.1
UNET D2 Smagorinsky Mixing=0
UNET D2 BCVolumeCheck=0
UNET D2 Cores=0
UNET D2 SolverType=PARDISO (Direct)
UNET D2 Minimum Iterations= 3
UNET D2 Maximum Iterations= 30
UNET D2 Restart Number= 10
UNET D2 Relaxation Coeff=1.3
UNET D2 SOR Precondition Iterations= 10
UNET D2 ILUT Maximum Fill= 8
UNET D2 ILUT Tolerance=1E-08
UNET D2 Convergence Tolerance=0.00001
UNET D1D2 MaxIter= 0
UNET D1D2 ZTol=0.01
UNET D1D2 QTol=0.1
UNET D1D2 MinQTol=1
Write IC File= 0
Write IC File at Fixed DateTime=0
Write IC File at Sim End=0
Echo Input=False
Echo Parameters=False
Echo Output=False
Write Detailed= 0
HDF Write Warmup=0
HDF Write Time Slices=0
HDF Flush=0
HDF Compression= 1
HDF Chunk Size= 1
HDF Spatial Parts= 1
HDF Use Max Rows=0
HDF Fixed Rows= 1
Calibration Method= 0
Calibration Iterations= 20
Calibration Max Change=0.05
Calibration Tolerance=0.2
Calibration Maximum=1.5
Calibration Minimum=0.5
Calibration Optimization Method= 1
WQ AD Non Conservative
WQ ULTIMATE=-1
WQ Max Comp Step=1HOUR
WQ Output Interval=15MIN
WQ Output Selected Increments= 0
WQ Create Restart=0
WQ Fixed Restart=0
WQ System Summary=0
WQ Write To DSS=0
Sorting and Armoring Iterations= 10
XS Update Threshold= 0.02
Bed Roughness Predictor= 0
Hydraulics Update Threshold= 0.02
Energy Slope Method= 1
Volume Change Method= 1
Sediment Retention Method= 0
Sediment TS Multiplier= 1
Warm Up Method= 0
XS Weighting Method= 0
Number of US Weighted Cross Sections= 1
Number of DS Weighted Cross Sections= 1
Upstream XS Weight=0
Main XS Weight=1
Downstream XS Weight=0
Number of DS XS's Weighted with US Boundary= 1
Upstream Boundary Weight= 1
Weight of XSs Associated with US Boundary= 0
Number of US XS's Weighted with DS Boundary= 1
Downstream Boundary Weight= 0.5
Weight of XSs Associated with DS Boundary= 0.5
Percentile Method= 0
Sediment Output Level= 3
Mass or Volume Output= 0
Output Increment Type= 1
Profile and TS Output Increment= 1
Transport Output Increment 1
XS Output Flag= 0
XS Output Increment= 10
Read HDF5 Sediment Hotstart= 0
Sediment Hotstart Type= 0
Write Gradation File= 0
Read Gradation Hotstart= 0
Write HDF5 File= 1
Write Binary Output= 1
Write DSS Sediment File= 0
DSS Sediment Output Type= 1
SV Curve= 0
Specific Gage Flag= 0
Subcell Erosion Methods= 0
Subcell Deposition Methods= 0
Advection Scheme= 1
Matrix Solver= 0
Implicit Weighting Factor= 1
Maximum Outer Loop Convergence Iterations= 5
Convergence Maximum Absolute= 0.001
Convergence RMSE= 0.0001
Grain Fractions Max Abs Error= 0.001
Max Subgrid Regions= 1
Max Subgrid Length Scale= 3.402823E+38
Initial Layer Thickness= 3.402823E+38
Min Layer Thickness= 3.402823E+38
Max Layer Thickness= 3.402823E+38
Number of Layers= 5

--- TENMILECK.f01 (steady flow) ---

Flow Title=Flows
Program Version=6.31
Number of Profiles= 1
Profile Names=01pct
River Rch & RM=TENMILECK,Main,20290
     415
River Rch & RM=TENMILECK,Main,15932
     463
River Rch & RM=TENMILECK,Main,12830
     546
River Rch & RM=TENMILECK,Main,12214
     627
River Rch & RM=TENMILECK,Main,10270
     698
River Rch & RM=TENMILECK,Main,4987
     790
River Rch & RM=TENMILECK,Main,3490
    1590
Boundary for River Rch & Prof#=TENMILECK,Main            , 1
Up Type= 0
Dn Type= 3
Dn Slope=0.00709
DSS Import GetInterval= 0
DSS Import GetPeak= 0
DSS Import FillOption= 0

--- TENMILECK.g01 (geometry) ---

Geom Title=Geometry
Program Version=6.31

River Reach=TENMILECK       ,Main
Reach XY= 30
2207194.65525668 679268.63977349     2207669.472      679939.564
     2207800.106      680690.486      2208722.24      681351.811
      2208811.58      681726.686     2208807.917      682385.807
     2208410.522      682598.141     2208584.223      683631.621
     2208477.255      684106.739     2207889.932      685338.475
     2207564.535      685283.703     2207143.302      685532.351
     2206717.633      685377.593      2206620.71      685513.235
     2205313.828      685233.481     2204795.843      684947.403
     2204448.497      684631.249     2204482.293      684458.006
     2203137.523      683589.527     2203372.149      683359.737
     2203097.059      683074.947     2203396.759      682937.474
      2203232.73      682517.213     2202929.596      682334.898
     2202770.747      682442.525     2202283.181      682026.414
     2201630.985      682148.606     2200619.796        683390.9
     2200136.637      683498.441     2199759.816      683069.939

Type RM Length L Ch R = 1 ,20290   ,458.7,436.9,439.5
XS GIS Cut Line= 3
 2206930.9643152679408.186896529 2207317.3241762 679235.69579858
2207422.34117572679197.646161074
#Sta/Elev= 30
       0 2060.24    27.6 2047.47    36.4 2044.82    56.4 2037.16      67 2034.66
   102.1 2028.65     124 2022.92   157.6 2016.81   172.8 2011.54   176.5 2009.81
   184.9 2004.63   189.7 2003.37   194.1 2002.88   202.8 2005.16   212.2 2004.82
     216 2004.12   227.3 1998.46   233.5 1997.62   345.4 1997.63   356.1 1998.37
   373.7 2002.71   384.8  2006.3   399.9 2008.72   430.3 2009.88   438.9 2009.29
   461.7 2011.57   472.9 2010.84   494.2 2012.63   512.7 2016.64   534.8 2025.27
#Mann= 5 ,-1,0
       0     .06       0     110     .05       0   227.3    .045       0
   356.1    .025       0  533.12      .1       0
Bank Sta=227.3,356.1
XS Rating Curve= 0 ,0
Exp/Cntr(USF)=0,0
Exp/Cntr=0.3,0.1

Type RM Length L Ch R = 1 ,19853   ,312.3,341.6,637.1
XS GIS Cut Line= 3
2207134.37812662679834.6530188912207722.65499709679484.692114924
2207768.95106991679359.360131863
#Sta/Elev= 30
       0 2059.13    39.3 2042.09    62.6 2028.96    71.9 2024.99    84.1 2021.53
   104.5  2018.2   116.2 2015.25   154.1 2000.09   160.3 1998.11     165 1997.63
   463.5 1997.62   472.91998.208   500.1 2009.19   521.8 2016.17   533.5 2019.01
   545.2 2020.36   551.3 2021.87   574.4 2020.48   588.5 2020.97   605.3 2023.96
   644.4 2027.03   652.3 2028.11   667.7 2032.19   688.2 2035.33   726.6 2038.27
   739.4 2039.72   747.6 2041.12   773.5 2047.35   777.8 2047.81   818.1 2047.65
#Mann= 6 ,-1,0
       0     .06       0     100     .07       0     110     .05       0
   160.3    .045       0   472.9    .025       0     680      .1       0
Bank Sta=160.3,472.9
XS Rating Curve= 0 ,0
Exp/Cntr(USF)=0,0
Exp/Cntr=0.3,0.1

Type RM Length L Ch R = 1 ,19511   ,303.5,356.8,557.4
XS GIS Cut Line= 3
     2207286.568      680086.797     2207659.305      679917.216
2208322.38651954679615.801276243
#Sta/Elev= 30
       0 2063.76    10.6 2063.71    19.3 2062.83    32.5 2058.96    45.7 2053.87
    72.1 2042.96      90 2034.57   102.1 2029.32   107.2 2026.88   120.2 2019.33
   129.2 2014.69   164.4 1998.34   165.5 1998.03   168.6 1997.63   959.7 1997.62
   962.4 1997.76   972.9 1998.59   981.7 1999.66    1008  2004.6  1016.8 2005.92
  1038.8 2005.53  1060.7 2006.32  1071.7  2007.3  1078.3 2007.43  1092.9 2008.36
  1095.9 2008.84  1109.1 2012.03  1117.9 2010.72  1126.7 2012.42  1137.9 2012.85
#Mann= 6 ,-1,0
       0     .05       0      20     .06       0      40     .03       0
     150     .05       0   165.5    .045       0   962.4    .025       0
Bank Sta=165.5,962.4
XS Rating Curve= 0 ,0
Exp/Cntr=0.3,0.1

Type RM Length L Ch R = 1 ,19154   ,405.5,369.7,480.8
XS GIS Cut Line= 2
2207284.52085596680321.6027773932208295.75013328680192.163055903
#Sta/Elev= 30
       0 2052.55     3.7 2053.44      40 2052.97   108.5  2057.6   124.7 2056.73
   193.1 2040.55   201.3 2039.07   216.5 2037.92   229.5 2034.36   261.8 2020.47
   275.3 2011.58   285.8 2006.25   302.1 1999.26   307.81997.956   310.2 1997.62
   770.31997.949     782 2002.12   810.2 2006.79   830.4 2014.33   874.7 2013.23
   893.8  2020.2     911  2022.4   923.1 2026.88   936.7 2024.72   951.4 2027.88
   963.5 2032.26   971.5 2034.22   999.7  2037.4  1011.9 2037.97  1019.5 2039.77
#Mann= 6 ,-1,0
       0     .05       0     140     .06       0     240      .1       0
   307.8    .045       0   770.3    .025       0     930     .03       0
Bank Sta=307.8,770.3
XS Rating Curve= 0 ,0
Exp/Cntr=0.3,0.1

Type RM Length L Ch R = 1 ,18785   ,641.3,639,637.4
XS GIS Cut Line= 4
2207464.86448645680769.4598030982207760.83987898680642.078383982
2208170.53128903680459.4257197172208248.29240342680426.422970929
#Sta/Elev= 30
       0 2030.93     3.6 2030.02    12.3 2025.67    71.5 2005.12      82 2003.64
    99.4 2003.04   132.2 1997.88   172.7  1997.7   345.71997.964   360.9 1997.95
   432.5 1997.83   495.1 1998.98   530.7  1997.8   585.9 1998.72   613.2 1998.62
   619.1  1997.9   625.3  1998.6   733.2  1998.2   746.5 1999.94   763.8 2005.85
   781.3 2007.47   785.6 2008.93     790  2012.1   798.6 2019.96   804.3 2023.23
   810.4 2023.93   820.4 2023.37   833.4 2024.05   846.4 2027.44   855.3 2027.86
#Mann= 7 ,-1,0
       0     .06       0      10     .05       0     260     .03       0
   345.7    .045       0   360.9     .03       0  742.22    .025       0
  810.79     .03       0
Bank Sta=345.7,360.9
XS Rating Curve= 0 ,0
Exp/Cntr(USF)=0,0
Exp/Cntr=0.3,0.1

Type RM Length L Ch R = 1 ,18146   ,116.3,131.3,104.4
XS GIS Cut Line= 3
2208022.28960122681227.6325401272208279.63647056681011.671851043
2208514.11142341 680824.30079321
#Sta/Elev= 30
       0 1972.84    14.4 1974.72    28.7 1972.89    54.7 1965.93    91.1 1962.25
   103.4 1959.79   164.3 1957.69   247.9 1957.58   284.2 1956.27   290.1 1955.66
   297.91952.496     304 1950.96   310.5  1952.4   315.8 1954.17   326.2  1952.3
   341.8 1952.31   366.6 1960.73   372.3 1962.01   384.8  1962.5   391.2 1963.92
   440.6 1977.36   461.7 1979.46   485.1 1983.63   519.4 1994.67   534.5 2000.79
   551.6 2003.87   564.2 2007.56   582.4 2013.78   597.1 2020.08   636.1 2034.78
#Mann= 8 ,-1,0
       0     .05       0     120     .03       0     260     .05       0
   297.9    .045       0   310.5     .05       0  375.96      .1       0
  415.96     .07       0  495.96      .1       0
Bank Sta=297.9,310.5
XS Rating Curve= 0 ,0
Exp/Cntr(USF)=0,0
Exp/Cntr=0.3,0.1

Type RM Length L Ch R = 1 ,18015   ,153.3,157.7,188.6
XS GIS Cut Line= 2
2208174.20711394681321.3034053082208511.95215026680861.594883652
#Sta/Elev= 30
       0 1984.19    15.8 1982.08    34.9  1978.1    44.8 1978.66    49.8 1976.64
    59.7 1968.82    64.7 1966.55    74.6 1966.36    84.5 1969.53   119.3 1953.42
   124.2 1951.95     154 1951.93   164.6 1950.23   178.8 1950.03     279 1951.56
   333.4 1950.06   339.1 1950.36   344.9 1951.93   362.5 1957.66   377.4 1965.57
   404.9 1966.49   408.7 1967.99   422.1 1976.19   449.2 1983.42   461.8  1988.5
   479.3 1997.82     510 2000.95   516.8 2002.47   531.2 2007.51   570.4 2023.22
#Mann= 7 ,-1,0
       0     .08       0      60      .1       0      80     .03       0
     154    .045       0   344.9      .1       0     390    .025       0
     450      .1       0
Bank Sta=154,344.9
XS Rating Curve= 0 ,0
Exp/Cntr(USF)=0,0
Exp/Cntr=0.3,0.1

Type RM Length L Ch R = 1 ,17857   ,103,63.8,72.3
XS GIS Cut Line= 3
2208301.02905881681347.2340450382208364.84828009681249.510862455
2208530.37938528681035.616753639
#Sta/Elev= 30
       0 1982.11      12 1977.57    21.6 1971.67    26.3  1970.4    31.1 1970.65
    35.9 1968.82      55 1960.59    70.2 1952.98    78.9 1951.59   102.8 1950.42
   122.2 1953.28   167.7  1952.9   176.4 1952.25   182.9 1950.28   187.9 1949.39
   198.1 1948.97   208.2 1949.36   213.2 1950.17   219.1 1952.09   224.8 1953.03
   264.7 1953.71   305.2 1957.32   311.7  1958.4   334.6 1965.91   350.3 1967.46
     356 1968.95   359.9  1970.9     370 1978.13   375.1 1980.42   387.2 1987.67
#Mann= 3 ,-1,0
       0      .1       0   182.9    .045       0   213.2      .1       0
#XS Ineff= 2 , 0
          142.65 1959.65
Permanent Ineff=
       F       F
Bank Sta=182.9,213.2
XS Rating Curve= 0 ,0
Exp/Cntr(USF)=0,0
Exp/Cntr=0.3,0.1

Type RM Length L Ch R = 1 ,17793   ,163.9,163.3,167.6
XS GIS Cut Line= 5
2208325.10946037681378.6990042592208392.95842632681288.444164082
2208450.48125832681243.471768158 2208494.3221328681162.004040148
2208559.28240838681064.730454314
#Sta/Elev= 30
       0 1987.46     6.9 1983.39    11.8 1981.28    41.9 1970.87    51.9 1965.65
    56.9 1964.58    63.3 1963.94     107 1952.12     112 1951.09   147.5 1948.83
   163.7 1949.11   170.2 1948.77   177.9 1948.12   197.6 1944.02   211.2 1943.54
   224.9 1944.41     234  1942.8   252.1 1942.33   261.2 1942.75   277.5  1945.8
   296.2 1951.69   310.6  1954.5   326.5 1958.69   346.8 1965.09   361.2 1971.22
     366 1972.14   375.6 1972.84   380.4 1975.45   387.1 1981.17   395.4 1986.43
#Mann= 4 ,-1,0
       0     .05       0      30      .1       0     234    .045       0
   261.2      .1       0
Bank Sta=234,261.2
XS Rating Curve= 0 ,0
Exp/Cntr=0.3,0.1

Type RM Length L Ch R = 1 ,17630   ,455.6,478.9,477.5
XS GIS Cut Line= 3
2208442.91730962681513.296331092 2208637.5182432681223.328052583
2208683.91316776681161.468153168
#Sta/Elev= 30
       0 1988.08     3.9 1986.73     9.4 1986.56    19.4 1989.49      29 1989.61
    33.9 1988.92    43.5 1986.08    53.1 1980.21    81.2 1969.44   107.7 1960.08
   116.3 1956.23   127.8 1954.27   138.6 1950.24   159.5 1944.42     188 1941.97
   202.8 1942.03   230.2 1940.07   237.4  1939.4   245.8 1939.43   254.7 1940.19
     272 1940.38   283.5 1942.01   296.6 1941.09   300.8 1941.61   322.9 1950.02
   346.9 1958.08   396.9 1972.41   415.5 1980.67   420.3 1981.74   426.5 1980.93
#Mann= 4 ,-1,0
       0     .08       0     110      .1       0   230.2    .045       0
   254.7      .1       0
Bank Sta=230.2,254.7
XS Rating Curve= 0 ,0
Exp/Cntr(USF)=0,0
Exp/Cntr=0.3,0.1

Type RM Length L Ch R = 1 ,17151   ,184.2,188.3,195.2
XS GIS Cut Line= 3
2208617.13712467681670.448684867 2208811.6130497681602.804884856
2209015.48394696 681540.79806818
#Sta/Elev= 30
       0 1992.91     6.5 1993.59    11.7  1992.6    24.4 1985.71    32.9 1981.79
    92.2 1960.59   119.6 1947.84   134.5 1941.71   138.5 1940.68     143 1940.28
   151.4 1941.93   155.7 1942.05   165.71938.971   189.6 1938.01     198 1938.74
   202.3 1940.59   210.7 1945.38     219 1947.53   252.5 1947.18   256.7 1946.24
   260.8 1944.64   277.6 1941.14   340.3 1941.73   365.4 1941.24   371.2 1941.49
   386.3 1943.99   398.8 1949.64   407.2 1951.88   411.4 1952.48     419 1951.79
#Mann= 4 ,-1,0
       0      .1       0   165.7    .045       0     198      .1       0
   395.9    .025       0
Bank Sta=165.7,198
XS Rating Curve= 0 ,0
Exp/Cntr(USF)=0,0
Exp/Cntr=0.3,0.1

Type RM Length L Ch R = 1 ,16962   ,145.9,149.7,150.6
XS GIS Cut Line= 3
2208642.66149289681802.1174807722208837.86813798681791.678622746
2209048.73307011681771.844792496
#Sta/Elev= 30
       0 1990.09     5.5 1990.45     9.5 1989.65    13.5 1987.64    25.5 1980.01
    33.6 1975.48    45.6 1973.27    53.6 1969.84    81.6 1959.77    93.6 1954.59
   121.7 1941.03   129.7 1938.02   141.7 1934.81   146.8 1932.22   149.7  1931.2
   153.7 1930.98   161.51932.095   173.4 1933.27   181.8 1933.13   196.2 1935.29
   203.6 1937.87   217.9 1944.75   221.9 1945.22   229.9 1945.19     234 1944.39
     242 1941.69     246 1941.15   394.7 1941.01   398.7 1942.06   407.3  1946.5
#Mann= 3 ,-1,0
       0      .1       0   146.8    .045       0   161.5      .1       0
Bank Sta=146.8,161.5
XS Rating Curve= 0 ,0
Exp/Cntr(USF)=0,0
Exp/Cntr=0.3,0.1

Type RM Length L Ch R = 1 ,16813   ,183.3,184.3,174.4
XS GIS Cut Line= 2
2208639.52983548681916.9449190622208972.52940652681947.217607338
#Sta/Elev= 30
       0 1969.09     4.7 1968.22    16.7 1967.72    20.7 1966.99    24.7 1965.52
    36.8 1959.03    44.8 1955.97    72.9    1946      93 1939.74   105.1 1937.12
   129.2 1933.35   137.2 1932.47   148.1 1930.35   153.3 1929.49   157.3 1929.25
   165.3 1929.31   172.8 1930.44   181.4 1932.42   185.4 1934.33   193.4 1939.09
   197.5 1940.35   217.5 1944.74   225.4 1945.28   233.6 1945.06   245.7 1943.55
   249.7 1943.87   261.7 1946.06   293.9 1949.54     326 1951.21   334.4 1952.35
#Mann= 3 ,0,0
       0      .1       0   148.1    .045       0   172.8      .1       0
Bank Sta=148.1,172.8
XS Rating Curve= 0 ,0
Exp/Cntr(USF)=0,0
Exp/Cntr=0.3,0.1

Type RM Length L Ch R = 1 ,16628   ,226.1,242.8,255.7
XS GIS Cut Line= 3
2208576.11672352682045.176266065 2208700.7102052682093.683618464
2208901.18699549682086.166731082
#Sta/Elev= 30
       0 1978.96     4.4  1976.6     8.6 1974.76    38.7 1963.56    51.6 1958.38
    64.4 1953.72    77.3 1948.56    81.6 1945.74    85.9 1942.15    90.2 1940.19
   111.7 1936.25   121.3 1935.05   133.1 1934.23   145.2 1932.32   157.2 1931.54
   164.61929.751   173.2 1929.27   186.7 1929.77   197.2 1930.46   213.2 1930.14
   229.2 1930.38   233.2 1930.75   241.2 1933.84   249.2  1937.8   253.2 1939.05
   265.3 1942.02   269.3 1942.71   278.2 1943.38   305.3 1943.88   334.3 1945.85
#Mann= 3 ,-1,0
       0      .1       0   164.6    .045       0   186.7      .1       0
Bank Sta=164.6,186.7
XS Rating Curve= 0 ,0
Exp/Cntr(USF)=0,0
Exp/Cntr=0.3,0.1

Type RM Length L Ch R = 1 ,16386   ,190.7,205.4,223.9
XS GIS Cut Line= 3
2208594.87958442682241.2243683322208693.80864194682263.208603335
2208940.70851197682321.551380844
#Sta/Elev= 30
       0  1946.5     4.4 1945.69    14.5 1944.71    21.8 1943.09    33.4 1941.36
    46.4 1938.76    62.8 1936.78    83.3 1933.48   103.8 1932.16   114.9 1932.51
   124.3 1931.09   144.9 1929.47   162.1 1929.38   190.1 1929.86   194.7 1929.44
   198.3 1929.16   244.6 1929.43   251.7 1929.86   255.8 1931.12   264.1 1936.02
   276.4 1941.12   288.7 1948.01   292.8 1949.62     297 1950.71   329.8 1952.44
   333.9 1952.88   338.1 1953.84   342.2 1955.22   350.4 1958.58     355 1960.07
#Mann= 3 ,0,0
       0      .1       0   194.7    .045       0   244.6      .1       0
Bank Sta=194.7,244.6
XS Rating Curve= 0 ,0
Exp/Cntr(USF)=0,0
Exp/Cntr=0.3,0.1

Type RM Length L Ch R = 1 ,16180   ,145.3,140.7,134.2
XS GIS Cut Line= 4
2208640.05745949 682335.549977062208705.22481826682416.598748794
2208742.92294883682486.9030884912208845.52911974682522.166364295
#Sta/Elev= 30
       0 1932.73     7.2 1931.11    12.4 1930.44    19.3 1930.19    26.8 1929.43
    35.4 1929.53    48.3 1929.17     104 1929.16   109.2 1929.07   113.7 1928.48
   118.3 1928.18   127.3 1928.06   136.2 1927.69     141 1927.78   143.51928.035
     150 1928.96   159.1 1929.69   163.7 1929.62   168.2 1929.13   172.7 1929.25
   177.3 1929.79   190.8 1933.37   214.9 1938.85   227.2 1942.41     240 1945.76
   248.5 1947.36   252.8 1947.88   261.2  1948.3   284.1 1948.18   292.3 1947.89
#Mann= 3 ,-1,0
       0      .1       0   127.3    .045       0   143.5      .1       0
Bank Sta=127.3,143.5
XS Rating Curve= 0 ,0
Exp/Cntr=0.3,0.1

Type RM Length L Ch R = 1 ,16040   ,109.9,107.9,105.4
XS GIS Cut Line= 4
2208508.12921426 682384.796339122208582.73066891682495.975498716
2208644.00759563 682543.856978042208747.43037451682554.635427117
#Sta/Elev= 30
       0 1940.91     5.3 1939.65    10.1 1937.98    20.5 1935.36    29.1 1932.23
    53.4 1927.12    64.7 1925.99    98.3 1925.36   112.7 1923.77   125.7 1923.14
   135.8 1923.75   140.8 1923.11   147.2 1921.49   152.9 1920.96   161.4 1921.01
   164.3 1921.53     170  1922.7   172.8 1922.96   189.9 1922.66   201.3 1922.99
   207.3 1924.03   211.8  1924.2   215.8 1923.69   219.9 1923.82     244 1925.25
     252 1926.26   271.3 1927.27   288.2 1931.63   300.3  1933.1   315.6 1936.44
#Mann= 3 ,-1,0
       0      .1       0   147.2    .045       0   164.3      .1       0
Bank Sta=147.2,164.3
XS Rating Curve= 0 ,0
Exp/Cntr(USF)=0,0
Exp/Cntr=0.3,0.1

Type RM Length L Ch R = 1 ,15932   ,141.4,139.7,136.9
XS GIS Cut Line= 4
2208456.87585733682486.7293517672208491.14474881682519.338651444
2208546.58729839682550.6830972752208682.72044592682607.757553536
#Sta/Elev= 30
       0 1930.94    12.6 1928.07    18.2 1926.55      21    1926    26.7 1925.44
    49.4 1919.66    58.2 1918.27      67 1917.63    71.5 1916.85    75.8 1916.02
    80.7 1915.56    91.7 1916.82   103.6  1918.1   108.2 1918.77   117.2 1920.68
   120.2 1920.83   138.7 1919.09   143.1 1919.31   147.4 1920.27   151.8 1920.88
   156.1 1920.94   164.8 1920.53   175.2 1920.61   186.5 1921.24   200.2  1921.3
   221.3 1922.04   227.2 1922.48   242.8 1924.54   251.5  1925.4   258.6 1926.63
#Mann= 3 ,-1,0
       0      .1       0    71.5    .045       0    91.7      .1       0
Bank Sta=71.5,91.7
XS Rating Curve= 0 ,0
Exp/Cntr=0.3,0.1

Type RM Length L Ch R = 1 ,15792   ,184.8,184.9,181.6
XS GIS Cut Line= 3
2208300.77011045682552.1785037992208491.55635023682617.144285664
2208628.55025248682661.786513075
#Sta/Elev= 30
       0 1949.09     3.5 1947.97      12 1946.24    24.7 1942.69      90 1925.84
    92.3 1925.08    96.6 1922.71   104.3 1916.62   106.4 1915.57   109.2 1914.41
   117.7 1914.12   121.9 1914.45   127.2 1915.48   134.6 1916.53   138.8 1916.73
   159.9 1916.41   176.8 1916.62     198 1918.07   206.4 1917.85   217.9    1917
   227.5 1917.22   235.9 1916.03   240.1 1915.91   252.8 1917.24   261.1 1917.47
   277.9 1916.99   303.6 1917.59   316.3 1918.52   336.8 1918.34   345.6  1918.7
#Mann= 3 ,-1,0
       0      .1       0   106.4    .045       0   127.2      .1       0
#XS Ineff= 2 , 0
                          266.99         1921.62
Permanent Ineff=
       F       F
Bank Sta=106.4,127.2
XS Rating Curve= 0 ,0
Exp/Cntr(USF)=0,0
Exp/Cntr=0.3,0.1

Type RM Length L Ch R = 1 ,15607   ,125.8,117.2,108.1
XS GIS Cut Line= 3
2208302.30566646  682705.45956342208584.63397676 682767.09997616
2208619.63964326682773.948910911
#Sta/Elev= 30
       0 1930.63    10.1 1927.96    18.3 1926.24    42.9 1921.95    75.6 1917.36
   104.3 1914.59   112.5 1913.37   120.6 1913.22   128.8  1912.6   141.1 1913.58
   145.8 1913.52   154.7 1912.42   161.6 1911.26   165.7 1911.22   169.8 1911.45
   172.7 1912.39     178  1913.7   182.1 1913.92   194.3 1913.52   206.3 1913.73
     223 1913.16   236.6 1914.08   251.7 1914.16   266.8 1915.68   276.2 1915.44
     289 1916.29   300.7 1915.61   304.8 1915.76     313 1916.74   324.6 1916.73
#Mann= 3 ,-1,0
       0      .1       0   154.7    .045       0   172.7      .1       0
Bank Sta=154.7,172.7
XS Rating Curve= 0 ,0
Exp/Cntr=0.3,0.1

Type RM Length L Ch R = 1 ,15490   ,89.5,93.6,97.6
XS GIS Cut Line= 4
2208354.18332457682886.5189951472208457.28315693682862.032784961
2208538.47427491682824.6590957312208611.93290547682809.194120877
#Sta/Elev= 30
       0 1922.23    18.5 1922.37    26.7 1921.83    59.6 1916.38    71.9 1913.68
      76 1912.36    80.2 1911.31    92.5 1910.16   100.7    1910   109.2 1910.68
   113.6 1910.69   120.9 1910.32   131.2 1910.38     140  1909.5     145 1909.17
   148.8 1909.17   153.2  1909.5     162 1910.86   178.1 1912.39   188.4 1912.69
   205.3 1912.02   209.3 1912.09   217.5 1913.29   225.7 1912.62   233.9 1912.99
     238 1913.55   246.1  1914.1   258.4  1915.5   266.6 1915.98   270.4    1916
#Mann= 3 ,0,0
       0      .1       0     140    .045       0   153.2      .1       0
Bank Sta=140,153.2
XS Rating Curve= 0 ,0
Exp/Cntr(USF)=0,0
Exp/Cntr=0.3,0.1

Type RM Length L Ch R = 1 ,15396   ,116.8,151.2,123.4
XS GIS Cut Line= 4
2208386.02595604682938.1818055752208475.37064651682938.181805575
2208504.17975078682933.4410668972208701.46741423682977.566403823
#Sta/Elev= 30
       0 1921.09    10.1 1920.44    26.1 1917.88    46.1  1913.8    66.1 1908.03
    70.1 1907.38    86.1 1907.55    97.2 1906.75   102.3 1905.95   106.4 1905.99
   110.4 1906.81   114.5 1907.53   130.8 1906.02   143.1 1906.77   147.2 1906.45
     154 1907.01   163.6 1908.92   171.8 1908.98     180 1909.85   192.3 1910.13
   204.6  1909.4   237.4  1911.4   242.3 1912.47   249.7 1915.73   253.8 1916.23
   270.2 1916.62   279.1  1919.8   290.7 1922.75   302.5 1927.11   320.7 1931.25
#Mann= 3 ,-1,0
       0      .1       0    97.2    .045       0   110.4      .1       0
Bank Sta=97.2,110.4
XS Rating Curve= 0 ,0
Exp/Cntr(USF)=0,0
Exp/Cntr=0.3,0.1

Type RM Length L Ch R = 1 ,15245   ,187.9,187.1,193.4
XS GIS Cut Line= 2
2208380.56182248683029.3602627912208659.42798711683079.233935955
#Sta/Elev= 30
       0 1918.11    40.2 1907.87    48.4 1906.02    64.6 1901.49    72.7 1900.01
    84.9 1901.34   101.2 1901.47   113.4 1900.62   121.5 1899.34   125.6  1899.1
   133.7 1899.15   141.8 1899.66     150 1899.16     154  1898.6     163 1896.18
   166.2 1895.63   171.9 1895.28   174.3 1895.36   178.4 1896.14   186.5 1898.23
   190.6 1900.29   202.6 1907.47     215 1912.39     219 1913.21   231.2 1913.58
   235.3 1914.76   247.5 1920.31   251.5 1921.79   271.8 1927.65   283.3 1930.62
#Mann= 3 ,-1,0
       0      .1       0     163    .045       0   178.4      .1       0
Bank Sta=163,178.4
XS Rating Curve= 0 ,0
Exp/Cntr(USF)=0,0
Exp/Cntr=0.3,0.1

Type RM Length L Ch R = 1 ,15058   ,240.9,231.4,223.2
XS GIS Cut Line= 3
2208366.40661583683188.775863241 2208545.8505853 683251.72217714
 2208608.7968992683243.266702138
#Sta/Elev= 30
       0 1912.12    10.4 1908.64    26.8 1904.19    55.1 1898.62      57 1898.07
    65.5 1894.39    69.7 1893.47    78.2 1893.55    90.9  1892.8   103.6 1892.69
   108.4 1892.03   114.7 1890.41   120.6 1889.86     129 1889.92   133.5 1890.46
   141.8 1894.71   142.9 1894.99     146  1895.5   158.6 1896.39     172 1898.88
   175.7    1900   184.1 1904.21   188.4 1906.02   204.6 1906.13   208.7 1906.72
   216.7 1911.63   232.9 1914.31   240.7 1916.38   247.9 1917.61   253.7 1919.13
#Mann= 3 ,0,0
       0      .1       0   114.7    .045       0   133.5      .1       0
Bank Sta=114.7,133.5
XS Rating Curve= 0 ,0
Exp/Cntr(USF)=0,0
Exp/Cntr=0.3,0.1

Type RM Length L Ch R = 1 ,14827   ,271.8,278.9,284.1
XS GIS Cut Line= 4
 2208246.3239413683464.183608199 2208456.1476328683462.031414888
2208572.82439782683435.5139682932208663.86763113683416.951755677
#Sta/Elev= 30
       0  1911.7    53.9 1907.42   141.9 1896.64   161.9 1893.55   185.9 1892.16
   189.9 1892.42   193.9 1893.48   197.9 1893.78   263.2 1894.93   267.3 1894.09
   275.5 1889.43   276.91889.076   279.6  1888.4   291.9 1888.35   300.1 1889.01
   304.2 1890.76   308.3 1893.34   312.4 1895.18   328.8 1898.28   332.9 1900.09
     337 1902.63     341 1904.27   369.6 1903.19   373.7 1903.22   377.8 1904.11
     386 1903.46   390.1 1905.02   394.1 1907.11   402.1 1910.11   422.4 1914.95
#Mann= 3 ,-1,0
       0      .1       0   276.9    .045       0   300.1      .1       0
Bank Sta=276.9,300.1
XS Rating Curve= 0 ,0
Exp/Cntr(USF)=0,0
Exp/Cntr=0.3,0.1

Type RM Length L Ch R = 1 ,14548   ,177.2,174.2,172.1
XS GIS Cut Line= 3
 2208292.3990657683663.0341450772208523.38106814683697.457018581
2208844.69443565683795.669783747
#Sta/Elev= 30
       0 1914.94    68.5 1909.16    88.7 1907.87   117.1 1908.22   173.7 1907.18
   191.8 1905.93   212.9 1903.13   234.4 1903.14   238.5 1902.67   246.3 1899.67
   271.41885.721   275.6 1884.31   278.8  1884.1     282 1884.48   285.2 1885.54
   288.4 1887.54   301.2  1897.5   305.5 1898.69   313.8 1897.73   322.2 1897.41
   359.8 1897.14   397.3  1899.1   410.5 1900.61     452 1907.08   472.8 1909.26
   502.1  1913.3     523 1914.93   535.5  1916.5   557.5  1917.2   569.5 1918.75
#Mann= 3 ,-1,0
       0      .1       0   271.4    .045       0   285.2      .1       0
Bank Sta=271.4,285.2
XS Rating Curve= 0 ,0
Exp/Cntr(USF)=0,0
Exp/Cntr=0.3,0.1

Type RM Length L Ch R = 1 ,14374   ,263.7,267.8,271.1
XS GIS Cut Line= 3
2208239.14204527683833.7164396912208560.14771305683880.287210147
2208869.51068822683933.510947811
#Sta/Elev= 30
       0  1947.2    17.2 1937.23    25.3 1934.08    45.5 1929.22    65.7 1926.23
      98 1917.91   110.2 1913.63   126.3 1910.37   170.8 1895.55   215.3 1891.09
   243.6 1890.11   257.2 1883.34   263.8 1881.09   267.8 1880.98   271.8 1881.42
   275.9 1883.28     288 1889.52   300.1  1891.4   312.3 1890.16   340.6  1889.5
   353.2 1893.45     365 1891.49   413.7 1891.04   454.3 1890.82   490.8 1892.35
   535.4 1899.72   551.7 1900.64   567.6 1899.92   580.1 1901.09   638.3 1913.86
#Mann= 5 ,-1,0
       0      .1       0   257.2    .045       0   275.9      .1       0
  464.37    .025       0  544.37      .1       0
Bank Sta=257.2,275.9
XS Rating Curve= 0 ,0
Exp/Cntr(USF)=0,0
Exp/Cntr=0.3,0.1

Type RM Length L Ch R = 1 ,14106   ,182.9,183.3,183.4
XS GIS Cut Line= 3
2208162.56773636684002.8921312442208574.29651391684183.177047501
2208832.11040091684281.283216892
#Sta/Elev= 30
       0 1987.89    19.2 1980.65    36.7 1975.23      76 1974.42    84.7 1969.37
   102.2 1955.39   119.7 1943.62   128.4 1938.92     159 1930.09   180.8 1925.79
   224.5 1909.16   241.9  1900.8   272.5 1888.12   294.3  1881.3   321.8 1875.12
   333.6  1874.1     338 1875.04   346.7 1879.65   355.2 1886.01   359.8 1887.91
   394.9 1886.41   498.6 1888.22   549.9 1891.12   626.1 1892.58   639.8 1893.52
   650.9 1895.42   665.5 1894.35   669.8 1895.01     704 1906.98   725.3 1913.03
#Mann= 5 ,-1,0
       0      .1       0   321.8    .045       0     338      .1       0
  539.47    .025       0  589.47      .1       0
Bank Sta=321.8,338
XS Rating Curve= 0 ,0
Exp/Cntr(USF)=0,0
Exp/Cntr=0.3,0.1

Type RM Length L Ch R = 1 ,13922   ,300.9,301.4,301.7
XS GIS Cut Line= 3
2208072.35797284684160.3616592712208508.13188804684354.292459229
 2208752.2565421684459.243245088
#Sta/Elev= 30
       0  1995.2     4.2 1992.74    15.6 1981.73    21.7 1977.41    41.4 1973.43
      61 1966.44    88.3 1966.67    94.4 1965.59   115.6 1956.86   174.9 1927.63
   227.7 1907.88   266.9 1897.22   288.3 1885.62     307 1879.06   327.7 1869.28
   336.5 1867.87   342.71869.569     358 1876.54   367.6  1882.5   371.9  1883.2
   398.2 1881.86   415.6 1879.41   586.1 1879.25   651.2 1880.82   658.9 1882.22
   668.6 1885.27   681.7 1886.84   690.4 1888.94   707.8 1895.12   742.7 1905.67
#Mann= 6 ,-1,0
       0      .1       0   327.7    .045       0   342.7      .1       0
     370     .03       0     470    .025       0  616.98      .1       0
Bank Sta=327.7,342.7
XS Rating Curve= 0 ,0
Exp/Cntr(USF)=0,0
Exp/Cntr=0.3,0.1

Type RM Length L Ch R = 1 ,13621   ,142.9,141.3,138.5
XS GIS Cut Line= 3
2208016.38399066684452.5137035492208275.37105241684580.681362091
2208471.60015721 684666.42110608
#Sta/Elev= 30
       0 1940.49    44.4 1921.63    62.2 1913.39    80.1 1906.21    89.9 1903.29
   110.8 1898.52   138.1 1890.88   174.8 1879.85   191.4 1872.56   206.3 1869.23
   224.3 1863.74   230.2 1862.81     245 1862.34   249.7 1862.69   254.1 1863.71
     272 1872.19     287 1871.38   320.2 1871.09   329.4 1869.66   337.9 1870.56
   364.1 1867.71   372.8 1865.74   381.5 1868.22   385.9 1868.51   410.1 1868.53
   442.6    1867   463.1 1868.04   481.9  1869.9     495 1870.37   503.1    1870
#Mann= 4 ,-1,0
       0      .1       0   224.3    .045       0   254.1      .1       0
  428.97    .025       0
Bank Sta=224.3,254.1
XS Rating Curve= 0 ,0
Exp/Cntr(USF)=0,0
Exp/Cntr=0.3,0.1

Type RM Length L Ch R = 1 ,13480   ,186.4,184.9,183.4
XS GIS Cut Line= 3
2207963.67994154684610.9566949882208231.50615215684704.651672956
2208455.13661843684790.391416946
#Sta/Elev= 30
       0 1925.86     4.8 1924.48    55.6 1904.76    72.6 1899.32    91.5 1890.68
   115.2 1881.74   131.9 1874.75   144.6 1871.27   165.4 1867.48   178.5 1867.87
   182.7  1866.2   195.5 1858.67   200.5 1856.33   208.2  1855.7   216.6 1856.25
   220.9 1857.53   233.6 1864.83   242.1  1867.7   246.3 1868.27   263.3 1867.12
   272.1 1868.23   278.4 1866.74     293 1861.53   297.3 1861.12   460.1 1860.95
   467.4 1861.95   481.5 1866.51   507.6 1867.98   515.8 1869.51   523.2 1871.92
#Mann= 5 ,-1,0
       0      .1       0   200.5    .045       0   216.6      .1       0
  293.74     .03       0  363.74      .1       0
Bank Sta=200.5,216.6
XS Rating Curve= 0 ,0
Exp/Cntr(USF)=0,0
Exp/Cntr=0.3,0.1

Type RM Length L Ch R = 1 ,13295   ,163,162.1,161.1
XS GIS Cut Line= 3
2207896.67822314684810.1467327832208186.60230591684870.252945065
 2208377.5279214684907.377370297
#Sta/Elev= 30
       0 1899.78    12.3  1900.3    19.1  1898.8    44.4 1882.79    49.5 1878.04
    52.6 1873.53    56.7 1865.78    60.8 1859.74    64.8 1857.76    83.3 1857.15
   109.8 1857.78     122 1860.69   127.3  1861.2   171.1 1861.71   179.2 1859.01
   193.41851.473   195.6 1850.48   199.7 1850.09   203.7 1850.37   207.8 1851.65
   211.9 1852.87   236.4 1863.48   240.5 1863.91     265 1863.24   289.7 1864.29
   375.1 1864.16   399.6 1863.29   415.9 1863.72   439.8 1866.05   490.6 1867.43
#Mann= 5 ,-1,0
       0      .1       0   193.4    .045       0   207.8      .1       0
  316.09     .03       0  416.09      .1       0
Bank Sta=193.4,207.8
XS Rating Curve= 0 ,0
Exp/Cntr(USF)=0,0
Exp/Cntr=0.3,0.1

Type RM Length L Ch R = 1 ,13133   ,116.1,116,115.8
XS GIS Cut Line= 2
2207819.83861712 684976.267044662208327.32155584685045.798441522
#Sta/Elev= 30
       0  1884.7    16.5 1877.21    20.5 1873.79    28.6 1863.07    33.1 1860.11
    52.8 1859.79    64.9 1858.78    85.1 1860.45     200 1861.04   210.3 1860.55
   218.4 1857.79   234.5 1850.63   238.71849.357   250.7 1848.24   258.81849.169
   275.4 1854.54     283 1858.53     287 1861.45     291 1863.04   299.1  1861.6
   311.2 1860.95   319.3 1861.32   331.3  1857.2   335.4 1856.82   375.8 1857.31
   468.7 1856.86   480.8 1857.17   488.9 1859.17     505 1865.04   512.2 1865.07
#Mann= 5 ,-1,0
       0      .1       0     180     .07       0     200      .1       0
   238.7    .045       0   258.8      .1       0
Bank Sta=238.7,258.8
XS Rating Curve= 0 ,0
Exp/Cntr(USF)=0,0
Exp/Cntr=0.3,0.1

Type RM Length L Ch R = 1 ,13017   ,115.1,114.8,115.7
XS GIS Cut Line= 5
2207806.43415781685018.2212437182208012.75951177685119.300626845
2208089.55019296685129.9025419972208159.72251636685146.720702151
2208313.52039178685134.345050387
#Sta/Elev= 30
       0 1875.51     1.9 1874.49     6.4 1870.01    10.8 1862.06    12.5  1860.2
    15.3  1857.9    18.5 1857.47   108.1 1857.37   131.1 1858.29   157.8 1857.24
   198.2 1857.98   215.7 1860.38   233.2 1860.23   241.3  1859.2   245.3  1857.7
   264.3 1847.82   269.9 1845.54   273.5 1845.74   278.51847.587   292.5 1854.85
   301.8 1860.62   305.9  1861.6     310 1860.54   359.3 1859.26   375.8 1860.12
   395.9 1858.43     420 1858.85   456.8 1861.68   492.2 1862.09   533.7 1865.39
#Mann= 10 ,-1,0
       0      .1       0      10     .08       0     120     .07       0
     190      .1       0  229.75     .07       0   264.3    .045       0
   278.5     .07       0  327.27      .1       0  429.43     .07       0
  529.43      .1       0
Bank Sta=264.3,278.5
XS Rating Curve= 0 ,0
Exp/Cntr(USF)=0,0
Exp/Cntr=0.3,0.1

Type RM Length L Ch R = 1 ,12902   ,64.5,71.4,79
XS GIS Cut Line= 4
2207750.32838804685098.5878252262207881.42214543685204.170137051
2208077.81526696685233.8166645172208253.75536991685191.792696473
#Sta/Elev= 30
       0  1869.4    94.8 1863.87   116.9 1861.89   120.5  1861.8   125.6  1862.5
   135.9 1859.78   157.2 1856.41   175.2 1854.75   196.2 1851.48   219.7 1848.59
     252 1846.72     263 1846.57   272.31843.589   280.3 1842.66   284.8 1843.41
   291.1 1847.58   296.5 1849.47   327.6    1857   336.8 1858.21   353.1 1857.56
   361.4 1857.97   373.5  1857.3   382.7 1855.58   398.2 1853.46   406.4 1852.75
   431.1 1852.62   451.6 1853.04   484.5 1856.17   524.6 1858.57   547.8 1861.27
#Mann= 5 ,-1,0
       0      .1       0   272.3    .045       0   284.8      .1       0
  406.94     .03       0  526.94     .07       0
Bank Sta=272.3,284.8
XS Rating Curve= 0 ,0
Exp/Cntr(USF)=0,0
Exp/Cntr=0.3,0.1

Type RM Length L Ch R = 1 ,12830   ,72.1,80.2,94.1
XS GIS Cut Line= 4
2207844.55473633685194.4954745612207917.61004034 685252.33092357
2208014.87371382685329.5503004852208067.55453694685439.177256528
#Sta/Elev= 30
       0 1860.78     4.3 1859.83     9.7 1858.29    15.9  1857.3    55.9 1852.57
    70.9 1850.48    86.2 1848.94   112.7 1847.31   116.9 1846.43     122 1844.84
   132.2 1841.17   139.6 1840.64   152.5 1841.03   153.4 1841.26   157.7 1842.73
   163.9  1846.8   166.8 1847.93   178.2 1849.28   183.3 1849.73     191 1849.16
   203.7 1849.71   234.7 1852.08   279.1 1851.73   292.4 1853.07   301.3 1852.83
   314.6 1854.24   327.9 1855.11   332.3 1855.98     335 1857.06     339 1858.29
#Mann= 6 ,-1,0
       0      .1       0   132.2    .045       0   153.4      .1       0
  163.18     .06       0  213.18     .07       0  297.37      .1       0
Bank Sta=132.2,153.4
XS Rating Curve= 0 ,0
Exp/Cntr(USF)=0,0
Exp/Cntr=0.3,0.1

Type RM Length L Ch R = 1 ,12750   ,56.2,58.8,61.9
XS GIS Cut Line= 4
 2207804.4829252685191.7778734752207869.08872321685281.355837037
2207907.36453597685353.2679701082207931.72187137685456.496677259
#Sta/Elev= 30
       0 1863.58    16.5 1862.41    36.3 1861.95    72.4 1861.98    95.4 1862.88
   100.4 1862.08   106.8 1859.75   115.6 1857.63   119.3 1855.69   130.3 1848.33
     134 1846.22   137.4 1845.25     142 1844.89   151.1  1843.4   158.31840.842
   164.6 1839.41   168.8 1839.28   177.7 1839.63   183.6 1840.82   195.9 1844.64
   204.1 1846.19   224.7 1847.04   232.4 1846.96     237 1847.41   257.6 1847.47
   261.7 1848.11   269.9 1851.76     274 1852.82   286.3 1853.59     298 1858.49
#Mann= 5 ,-1,0
       0      .1       0   119.8     .07       0   158.3    .045       0
   183.6     .07       0  231.27      .1       0
Bank Sta=158.3,183.6
XS Rating Curve= 0 ,0
Exp/Cntr(USF)=0,0
Exp/Cntr=0.3,0.1

Type RM Length L Ch R = 1 ,12691   ,53.5,60.1,67.1
XS GIS Cut Line= 3
2207774.40558683685231.8083189072207834.71898876685329.237660488
2207879.95404021685474.221799744
#Sta/Elev= 30
       0 1865.45    34.5 1863.87    58.1 1863.19    66.2 1862.46    72.2 1862.42
    79.4 1861.54      87 1858.87      91 1857.11    94.6 1855.12   100.4 1851.44
   105.1 1847.93   109.8 1845.72   114.6  1844.8   122.9  1842.6   127.1  1841.4
   133.51838.989   135.5 1838.34   139.7 1838.16     148 1838.55   149.41839.153
   152.2 1840.36   156.4 1842.77     169 1844.33   202.5 1844.89   210.9 1845.79
   240.3 1847.88   244.4 1849.16   246.6 1850.24     257 1856.26   266.5 1859.83
#Mann= 5 ,-1,0
       0      .1       0      80     .07       0   133.5    .045       0
   149.4     .07       0  184.59      .1       0
Bank Sta=133.5,149.4
XS Rating Curve= 0 ,0
Exp/Cntr(USF)=0,0
Exp/Cntr=0.3,0.1

Type RM Length L Ch R = 1 ,12631   ,150.9,151.4,151.7
XS GIS Cut Line= 4
2207745.49192188  685232.50493872207793.59417967685306.631269546
2207771.36391728685398.9815739192207752.42970225685489.001170862
#Sta/Elev= 30
       0 1860.92    11.1  1859.7    19.9 1857.43    29.4 1855.98    51.6 1851.52
    77.1 1849.29    88.4  1848.9    95.1 1844.56    98.3 1843.62   104.9 1842.84
   115.7 1839.79   123.9 1839.25   132.1 1838.06   136.2 1838.16   141.31839.143
   148.6 1842.04   152.7 1842.37   156.8  1841.8     165 1842.59   181.5  1842.9
   193.8 1842.23   204.8 1842.49   214.9 1841.81   238.7 1842.73   246.9  1841.4
   248.7 1841.46     251 1841.68   255.1 1842.88   267.4 1847.74   275.3 1849.04
#Mann= 5 ,-1,0
       0      .1       0      80     .07       0   123.9    .045       0
   141.3     .07       0  178.37      .1       0
Bank Sta=123.9,141.3
XS Rating Curve= 0 ,0
Exp/Cntr(USF)=0,0
Exp/Cntr=0.3,0.1

Type RM Length L Ch R = 1 ,12480   ,275.4,266.4,256.4
XS GIS Cut Line= 5
 2207659.1163043685235.0374466822207656.12058024685247.519630266
2207630.15763838685340.8863634742207684.03516211685478.309312164
2207660.74823053685597.665192283
#Sta/Elev= 30
       0 1857.11      27 1852.32    35.3  1850.3    39.5 1848.47    51.9 1840.73
    58.21838.097    60.2 1837.56    72.31838.024      81 1841.06    85.6 1841.95
   111.5 1841.68   122.9 1842.12   131.5 1841.53   148.7 1841.71   161.6 1840.99
   178.8 1841.81   191.8 1841.47   200.3 1842.09   216.5 1842.39   226.8 1843.12
   241.2 1843.57   257.4 1845.55   293.8 1842.12     301 1842.17   314.2 1844.08
   317.7 1845.15   325.5 1848.87   329.6 1849.62   349.9 1851.12     379 1854.17
#Mann= 6 ,-1,0
       0      .1       0    58.2    .045       0    72.3      .1       0
  169.75     .06       0  277.35      .1       0  377.35     .03       0
Bank Sta=58.2,72.3
XS Rating Curve= 0 ,0
Exp/Cntr(USF)=0,0
Exp/Cntr=0.3,0.1

Type RM Length L Ch R = 1 ,12214   ,102.5,94.4,80.1
XS GIS Cut Line= 4
2207396.19091917685214.742803476 2207394.3083454685340.307854729
 2207444.6226622685455.0374566362207480.46395142685569.801991126
#Sta/Elev= 30
       0 1875.86    30.4 1866.38    46.4 1862.08   102.4 1851.66   125.6 1845.35
   135.3 1844.14   139.8  1842.5     144  1840.1   148.4 1838.58   161.5 1837.87
   170.2 1838.22   176.81837.303   182.3 1836.44   196.4 1836.64     1991837.213
   205.1 1839.12   209.5 1839.84   213.9 1839.63   218.3 1838.41   221.8 1838.18
   231.4 1838.82   240.1 1838.56   261.8 1841.78   282.4 1842.91     303 1845.38
   316.1 1844.81   319.3 1845.13   338.4  1849.7   357.6 1852.87   371.1 1856.06
#Mann= 5 ,-1,0
       0      .1       0      90     .06       0   176.8    .045       0
     199      .1       0  290.86     .03       0
Bank Sta=176.8,199
XS Rating Curve= 0 ,0
Exp/Cntr(USF)=0,0
Exp/Cntr=0.3,0.1

Type RM Length L Ch R = 1 ,12119   ,46.1,41.8,40.8
XS GIS Cut Line= 5
2207222.99999915 685419.476106972207303.37920596685433.046622404
2207367.05623992685434.0905082072207415.65663716685424.938582769
2207472.56019095685590.461986402
#Sta/Elev= 30
       0 1840.29    13.4    1841    21.5 1839.25    25.5 1838.91    41.8 1838.94
    51.1 1838.47    70.2 1838.88   117.9 1836.22   122.3  1835.6     1281836.184
   130.3 1836.61   142.3 1836.96   162.6 1838.32   174.8  1838.1   191.1 1839.13
   194.9 1839.16   199.1  1838.2   203.4 1837.95   211.8 1838.59   220.3 1838.34
   228.7 1839.77   237.2 1840.33   262.6 1843.76   275.3 1844.34     296 1846.58
   304.9 1846.13     318 1849.34   334.5 1851.85   352.6 1856.48   369.7 1860.21
#Mann= 4 ,-1,0
       0      .1       0   117.9    .045       0     128      .1       0
  274.66     .03       0
Bank Sta=117.9,128
XS Rating Curve= 0 ,0
Exp/Cntr(USF)=0,0
Exp/Cntr=0.3,0.1

Type RM Length L Ch R = 1 ,12077   ,110.5,135,155.4
XS GIS Cut Line= 5
2207222.99999915685457.0559958652207293.98423373685472.714282905
2207364.96846831685473.7581687082207427.14764024685468.221561883
2207467.80294683685594.890682901
#Sta/Elev= 30
       0 1838.56      38 1837.62    46.3    1838    58.1 1837.84    66.7 1836.59
    70.8 1836.25    74.9 1836.78    78.9 1836.74    82.9 1836.03    90.9  1835.2
      95 1834.45    98.9 1834.16   110.9 1833.94   114.9 1834.13   122.6 1835.35
   130.9 1836.86   142.9 1838.58   154.9  1838.8   176.7 1839.85   203.9 1840.42
   232.3  1844.2   244.9 1844.67   264.9 1846.71   271.3  1846.4   274.5 1846.49
   282.7 1848.71   286.9 1849.59   303.1 1852.29   320.5 1856.97   339.1 1860.93
#Mann= 5 ,-1,0
       0      .1       0    90.9    .045       0   122.6      .1       0
  236.11     .03       0  336.11      .1       0
Bank Sta=90.9,122.6
XS Rating Curve= 0 ,0
Exp/Cntr(USF)=0,0
Exp/Cntr=0.3,0.1

Type RM Length L Ch R = 1 ,11942   ,109.3,113,116.6
XS GIS Cut Line= 3
2207183.74302547685452.5135615062207214.91646402685486.901611933
2207226.01173832685612.278211487
#Sta/Elev= 30
       0 1839.73    12.6 1839.31    20.6 1837.54    24.5 1837.01    27.9 1836.92
    33.3  1837.3    48.7 1836.51    56.7 1836.29    60.7 1835.62    64.8 1834.63
    68.8 1834.29    72.8 1834.18    76.31833.638    80.8 1833.14    92.9 1833.62
    96.9 1834.43   100.9 1835.05   104.9 1835.28   108.9 1836.01     113 1835.85
     121 1833.83     125 1833.71     129 1834.38   141.1 1835.96   149.1  1837.4
   157.1 1838.15   161.1 1838.67   165.2 1839.53   169.2 1841.11   172.3 1842.59
#Mann= 3 ,-1,0
       0      .1       0    76.3    .045       0    92.9      .1       0
Bank Sta=76.3,92.9
XS Rating Curve= 0 ,0
Exp/Cntr(USF)=0,0
Exp/Cntr=0.3,0.1

Type RM Length L Ch R = 1 ,11829   ,71.8,74,75.7
XS GIS Cut Line= 2
2207147.63671286685333.1749507192207087.15044283685618.876055973
#Sta/Elev= 30
       0 1849.42    12.3 1848.15    24.5 1845.85    36.8 1845.63      45 1843.26
    57.2 1841.43    65.4 1841.06    73.6 1839.89    85.9 1840.34      94 1840.16
   114.5 1838.32   118.6  1837.7   132.6  1834.2   143.1 1833.67   159.5 1834.52
   179.9 1834.82     184 1834.66     1901833.402   196.3 1832.96   204.31833.353
   212.6 1834.91   220.8  1835.5   224.9 1834.92   237.1  1834.9   253.5 1831.98
   257.6 1832.58   273.9 1837.48     278 1838.36   286.2 1839.46     292 1839.67
#Mann= 4 ,-1,0
       0     .06       0      70      .1       0     190    .045       0
   204.3      .1       0
Bank Sta=190,204.3
XS Rating Curve= 0 ,0
Exp/Cntr(USF)=0,0
Exp/Cntr=0.3,0.1

Type RM Length L Ch R = 1 ,11755   ,302.4,304.7,296.1
XS GIS Cut Line= 3
2207071.80312041 685333.200008322207054.05706177685461.597962045
2207000.81888583685599.390887994
#Sta/Elev= 30
       0 1846.83    16.1 1844.52    44.4 1838.67    56.5 1839.15    72.7 1838.71
    76.7 1837.67    80.7 1837.02    88.8 1836.46    96.9 1834.91   129.2 1834.23
   137.7 1832.16     142 1830.75   150.6 1827.12   154.9 1825.98   163.5 1824.68
     171 1826.06   172.1 1826.21   176.3 1825.69   180.6 1825.61   184.9 1827.15
   197.8 1828.34   209.5 1830.79   227.8 1835.42   232.1 1834.83     239 1832.64
   245.2 1831.11   249.2 1830.54   253.5  1832.1   262.1 1836.53   277.3 1837.81
#Mann= 4 ,-1,0
       0     .06       0      70      .1       0   154.9    .045       0
     171      .1       0
Bank Sta=154.9,171
XS Rating Curve= 0 ,0
Exp/Cntr(USF)=0,0
Exp/Cntr=0.3,0.1

Type RM Length L Ch R = 1 ,11451   ,289.7,300.3,298.2
XS GIS Cut Line= 2
 2206806.4469808685265.3580569822206754.89706462685577.235049871
#Sta/Elev= 30
       0  1834.6     5.3 1834.48      12 1833.19    24.1 1833.45    36.3 1832.49
    44.4 1832.66    48.5 1832.08    52.5 1829.87    60.6  1823.9    64.7 1821.23
    68.7 1819.66    72.8 1819.13    76.8 1819.07   105.2 1819.28   109.3 1819.02
   117.4 1816.68   125.5  1816.3   133.6 1816.73   149.8 1819.88   157.9 1820.99
   186.3 1820.91   210.6 1822.12   218.7 1821.96   222.8 1822.24   234.9 1824.59
     239 1824.73   255.2  1826.6   287.7 1832.69   303.9 1836.52   316.1 1840.81
#Mann= 4 ,-1,0
       0     .06       0      40      .1       0   117.4    .045       0
   133.6      .1       0
Bank Sta=117.4,133.6
XS Rating Curve= 0 ,0
Exp/Cntr(USF)=0,0
Exp/Cntr=0.3,0.1

Type RM Length L Ch R = 1 ,11150   ,229.9,230.6,224.8
XS GIS Cut Line= 3
2206652.83072123685149.7975342012206622.90102504685395.066898521
2206501.36549903685673.137002574
#Sta/Elev= 30
       0 1844.63    19.5 1837.35      88 1832.64    92.1 1832.07   100.1 1828.53
   176.7 1826.18   188.8 1824.87   208.9 1825.15   245.2 1821.38   275.6 1814.42
   296.3 1812.91   310.5 1813.03   338.9 1810.47   345.4 1809.59   358.5 1810.41
   363.8 1812.73   393.5 1834.99   406.5 1842.02   423.7 1845.58   457.3 1855.83
   467.7 1860.16     472 1861.16   489.5 1863.08     507 1863.03   521.1 1861.89
   524.2 1862.81   527.2 1864.86   541.9 1877.55   546.2 1879.84   550.6 1880.97
#Mann= 3 ,-1,0
       0      .1       0   338.9    .045       0   358.5      .1       0
Bank Sta=338.9,358.5
XS Rating Curve= 0 ,0
Exp/Cntr(USF)=0,0
Exp/Cntr=0.3,0.1

Type RM Length L Ch R = 1 ,10920   ,290.3,286.8,282.8
XS GIS Cut Line= 2
2206460.22858241685140.0969689862206363.32142212685480.433559714
#Sta/Elev= 30
       0 1833.68    21.9 1825.49    34.4 1822.91    46.9 1821.88    71.8 1821.12
    80.1 1818.69    88.5 1819.03   100.9 1818.56   113.4 1819.42   138.4 1818.51
     155 1817.35   169.3 1817.82     180 1815.94   195.2 1814.41   209.1 1811.99
   221.6 1809.39   227.81807.455   230.8 1806.84   237.2 1806.64   246.5 1806.73
   250.41807.266   271.5 1810.44   279.8 1813.83   292.2 1820.05   308.9 1827.56
   321.4 1832.57   325.5 1833.61   333.8  1834.6   342.2 1838.09   353.9 1841.43
#Mann= 4 ,-1,0
       0     .06       0      60      .1       0   227.8    .045       0
   250.4      .1       0
Bank Sta=227.8,250.4
XS Rating Curve= 0 ,0
Exp/Cntr(USF)=0,0
Exp/Cntr=0.3,0.1
